--- PECKSRNT4.prj (project) ---

Proj Title=PECKSRNT4
Current Plan=p01
Default Exp/Contr=0,0
English Units
Geom File=g01
Flow File=f01
Plan File=p01
BEGIN DESCRIPTION:
---------- MODELED AS PART OF WVEMD CTP PROGRAM, 2023----------
Stream Name: Pecks Run Tributary 4
Flood Zone:  AFH
Upshur County, WV
HEC-RAS Version: RAS 6.3
Vertical Datum: NAVD88
Projection: NAD 1983 StatePlane West Virginia S FIPS 4702 (US Feet)
Terrain: 1-meter LIDAR (FEMA Region III 3DEP collected 2016-2018)
Land Use: 2019 NLCD
Hydrologic Method:
WV SIR2010-5033 regression equations
Additional Model Notes:
None
END DESCRIPTION:
DSS Export Rating Curves= 0
DSS Export Rating Curve Sorted= 0
DSS Export Volume Flow Curves= 0
DXF OffsetX= 0
DXF OffsetY= 0
DXF ScaleX= 0
DXF ScaleY= 0

--- PECKSRNT4.p01 (plan) ---

Plan Title=Floodplain
Program Version=6.30
Short Identifier=Floodplain
Geom File=g01
Flow File=f01
Subcritical Flow
K Sum by GR= 0
Std Step Tol= 0.01
Critical Tol= 0.01
Num of Std Step Trials= 20
Max Error Tol= 0.3
Flow Tol Ratio= 0.001
Split Flow NTrial= 30
Split Flow Tol= 0.02
Split Flow Ratio= 0.02
Log Output Level= 0
Friction Slope Method= 1
Unsteady Friction Slope Method= 2
Unsteady Bridges Friction Slope Method= 1
Parabolic Critical Depth
Global Vel Dist= 0 , 0 , 0
Global Log Level= 0
CheckData=False
Encroach Param=-1 ,0,0, 0
Mapping Interval=1HOUR
Computation Time Step Use Courant=        0
Computation Time Step Use Time Series=    0
Computation Time Step Count To Double=0
Computation Time Step Max Doubling=0
Computation Time Step Max Halving=0
Computation Time Step Residence Courant=0
Run HTab= 0
Run UNet= 0
Run Sediment= 0
Run PostProcess= 0
Run WQNet= 0
Run RASMapper=-1
UNET Theta= 0
UNET Theta Warmup= 0
UNET ZTol= 0
UNET ZSATol= 0
UNET MxIter= 0
UNET Max Iter WO Improvement= 0
UNET MaxInSteps= 0
UNET DtIC= 0
UNET DtMin= 0
UNET MaxCRTS= 0
UNET WFStab= 0
UNET SFStab= 0
UNET WFX= 1
UNET SFX= 1
UNET Gravity=32.17405
UNET 1D Methodology=Finite Difference
UNET DSS MLevel= 1
UNET Pardiso=0
UNET DZMax Abort= 0
UNET Use Existing IB Tables= 0
UNET Froude Reduction=False
UNET Froude Limit= 0
UNET Froude Power= 0
UNET D1 Cores= 0
UNET WindReference=Eulerian
UNET WindDragFormulation=Hsu (1988)
UNET D2 Coriolis=0
UNET D2 Cores= 0
UNET D2 Theta= 1
UNET D2 Theta Warmup= 1
UNET D2 Z Tol= 0.01
UNET D2 Volume Tol= 0.01
UNET D2 Max Iterations= 20
UNET D2 Equation= 0
UNET D2 RampUpFraction=0.1
UNET D2 TimeSlices= 1
UNET D2 Turbulence Formulation=Non-Conservative (original)
UNET D2 Eddy Viscosity=0.3
UNET D2 Transverse Eddy Viscosity=0.1
UNET D2 Smagorinsky Mixing=0
UNET D2 BCVolumeCheck=0
UNET D2 Cores=0
UNET D2 SolverType=PARDISO (Direct)
UNET D2 Minimum Iterations= 3
UNET D2 Maximum Iterations= 30
UNET D2 Restart Number= 10
UNET D2 Relaxation Coeff=1.3
UNET D2 SOR Precondition Iterations= 10
UNET D2 ILUT Maximum Fill= 8
UNET D2 ILUT Tolerance=1E-08
UNET D2 Convergence Tolerance=0.00001
UNET D1D2 MaxIter= 0
UNET D1D2 ZTol=0.01
UNET D1D2 QTol=0.1
UNET D1D2 MinQTol=1
Write IC File= 0
Write IC File at Fixed DateTime=0
Write IC File at Sim End=0
Echo Input=False
Echo Parameters=False
Echo Output=False
Write Detailed= 0
HDF Write Warmup=0
HDF Write Time Slices=0
HDF Flush=0
HDF Compression= 1
HDF Chunk Size= 1
HDF Spatial Parts= 1
HDF Use Max Rows=0
HDF Fixed Rows= 1
Calibration Method= 0
Calibration Iterations= 20
Calibration Max Change=0.05
Calibration Tolerance=0.2
Calibration Maximum=1.5
Calibration Minimum=0.5
Calibration Optimization Method= 1
WQ AD Non Conservative
WQ ULTIMATE=-1
WQ Max Comp Step=1HOUR
WQ Output Interval=15MIN
WQ Output Selected Increments= 0
WQ Output face flow=0
WQ Output face velocity=0
WQ Output face area=0
WQ Output face dispersion=0
WQ Output cell volume=0
WQ Output cell surface area=0
WQ Output cell continuity=0
WQ Output cumulative cell continuity=0
WQ Output face conc=0
WQ Output face dconc_dx=0
WQ Output face courant=0
WQ Output face peclet=0
WQ Output face adv mass=0
WQ Output face disp mass=0
WQ Output cell mass=0
WQ Output cell source sink temp=0
WQ Output nsm pathways=0
WQ Output nsm derived pathways=0
WQ Create Restart=0
WQ Fixed Restart=0
WQ System Summary=0
WQ Write To DSS=0
Sorting and Armoring Iterations= 10
XS Update Threshold= 0.02
Bed Roughness Predictor= 0
Hydraulics Update Threshold= 0.02
Energy Slope Method= 1
Volume Change Method= 1
Sediment Retention Method= 0
Sediment TS Multiplier= 1
Warm Up Method= 0
XS Weighting Method= 0
Number of US Weighted Cross Sections= 1
Number of DS Weighted Cross Sections= 1
Upstream XS Weight=0
Main XS Weight=1
Downstream XS Weight=0
Number of DS XS's Weighted with US Boundary= 1
Upstream Boundary Weight= 1
Weight of XSs Associated with US Boundary= 0
Number of US XS's Weighted with DS Boundary= 1
Downstream Boundary Weight= 0.5
Weight of XSs Associated with DS Boundary= 0.5
Percentile Method= 0
Sediment Output Level= 3
Mass or Volume Output= 0
Output Increment Type= 1
Profile and TS Output Increment= 1
Transport Output Increment 1
XS Output Flag= 0
XS Output Increment= 10
Read HDF5 Sediment Hotstart= 0
Sediment Hotstart Type= 0
Write Gradation File= 0
Read Gradation Hotstart= 0
Write HDF5 File= 1
Write Binary Output= 1
Write DSS Sediment File= 0
DSS Sediment Output Type= 1
SV Curve= 0
Specific Gage Flag= 0
Subcell Erosion Methods= 0
Subcell Deposition Methods= 0
Advection Scheme= 1
Matrix Solver= 0
Implicit Weighting Factor= 1
Maximum Outer Loop Convergence Iterations= 5
Convergence Maximum Absolute= 0.001
Convergence RMSE= 0.0001
Grain Fractions Max Abs Error= 0.001
Max Subgrid Regions= 1
Max Subgrid Length Scale= 3.402823E+38
Initial Layer Thickness= 3.402823E+38
Min Layer Thickness= 3.402823E+38
Max Layer Thickness= 3.402823E+38
Number of Layers= 5

--- PECKSRNT4.f01 (steady flow) ---

Flow Title=Flows
Program Version=6.31
Number of Profiles= 1
Profile Names=01pct
River Rch & RM=PECKSRNT4,Main,2829
     134
River Rch & RM=PECKSRNT4,Main,1003
     150
Boundary for River Rch & Prof#=PECKSRNT4,Main            , 1
Up Type= 0
Dn Type= 3
Dn Slope=0.01239
DSS Import GetInterval= 0
DSS Import GetPeak= 0
DSS Import FillOption= 0

--- PECKSRNT4.g01 (geometry) ---

Geom Title=Geometry
Program Version=6.31

River Reach=PECKSRNT4       ,Main
Reach XY= 30
2197111.24299959750409.7486300682197206.41155076750666.143109527
2197222.42958039750678.0779005082197267.61800273750774.920679668
 2197277.2871625 750865.765808692197315.38564215750936.863480202
 2197322.9828122750974.3350119762197384.82714988750963.844161888
 2197413.6450689750977.5798058342197448.88915627751031.675381796
2197466.45193634 751083.69614943  2197378.120993751132.074353444
2197374.72214305751190.3724662882197384.71011717751336.589058926
2197397.91974433751411.0572536022197441.75688398751470.027476629
2197486.28677763751582.9594627832197502.93911474751674.126109238
2197511.14108184751730.2859728782197499.49874202751857.613369313
2197495.39586488752149.4864083292197487.34896608752171.404670261
 2197505.9869926752227.8133802982197500.81511645752253.672761085
2197515.13420396752300.204211011 2197506.8273052752325.150221033
2197589.90769051752497.3310416772197607.79003605752855.775137549
2197625.65652203752962.864055849     2197635.507      752976.742

Type RM Length L Ch R = 1 ,2829    ,88.2,88.2,88.2
XS GIS Cut Line= 3
2197049.54542405 750463.204182062197181.39249924750407.312487141
 2197209.3383467 750384.38256102
#Sta/Elev= 30
       0 1445.94     3.6 1444.93    15.9 1441.13    20.2 1440.09    24.9  1439.3
    28.9 1438.87    37.1 1438.57    55.4 1438.84    63.7  1438.7      68 1437.95
    72.11436.893    76.7 1436.29    78.31436.887    81.1 1437.96    85.4 1439.12
    95.1 1439.54   106.7 1439.56   116.4 1439.78   128.6 1440.38   133.2 1440.79
   137.8 1441.47   141.9 1442.39   143.9 1443.08   146.7 1444.25   152.4 1447.44
   155.2 1448.88   159.2 1450.76   162.3 1452.09   172.3 1455.47   179.4 1457.47
#Mann= 4 ,-1,0
       0     .06       0      40     .05       0    72.1    .045       0
    78.3     .05       0
#XS Ineff= 2 , 0
           52.85  1441.3
Permanent Ineff=
       F       F
Bank Sta=72.1,78.3
XS Rating Curve= 0 ,0
Exp/Cntr(USF)=0,0
Exp/Cntr=0.3,0.1

Type RM Length L Ch R = 1 ,2741    ,75.8,76.6,77.2
XS GIS Cut Line= 2
2197082.94931181 750547.807575542197251.62594747750467.716511127
#Sta/Elev= 30
       0 1449.94     5.8 1448.83    10.2 1447.84    14.6 1446.65    19.1 1445.25
    32.4 1440.28    36.8 1439.04    41.9 1438.28    54.5 1438.06    58.9 1437.52
    64.5 1436.44    68.9 1435.78    71.9 1435.84    73.91436.449    76.6 1437.33
      78 1437.36    81.1 1437.05    85.5 1436.11      87 1435.97    89.9 1435.78
      99  1435.6   103.2 1435.68   107.6 1436.16   116.5 1438.28   120.9 1438.91
     129 1440.81   138.6 1442.75   156.3  1446.9     171 1449.07   186.7 1452.06
#Mann= 3 ,-1,0
       0     .06       0    64.5    .045       0    73.9     .06       0
Bank Sta=64.5,73.9
XS Rating Curve= 0 ,0
Exp/Cntr(USF)=0,0
Exp/Cntr=0.3,0.1

Type RM Length L Ch R = 1 ,2664    ,104.5,104.5,104
XS GIS Cut Line= 3
2197109.09561235750613.6690117132197241.67372226750563.364551573
2197292.44831754750537.507118791
#Sta/Elev= 30
       0 1449.54       9 1447.61    15.2 1446.02    20.4  1444.4    33.2 1440.08
    36.9 1439.24    46.2 1437.93    58.9 1437.05    61.7 1436.73    63.2 1436.52
    66.91435.686      71  1435.1    71.7  1435.1    73.4 1435.65    80.3 1438.22
    84.6 1438.37    93.1 1438.05   110.2 1437.99   127.4 1437.41   131.6  1437.5
   135.5 1437.85   140.2 1438.41   144.6 1439.15   162.6 1442.75   167.1 1444.02
   171.5 1445.62     176 1447.07   192.9 1450.99   195.8 1451.85   198.8 1453.03
#Mann= 5 ,-1,0
       0      .1       0    66.9    .045       0    73.4      .1       0
    80.3     .06       0   192.9     .05       0
Bank Sta=66.9,73.4
XS Rating Curve= 0 ,0
Exp/Cntr(USF)=0,0
Exp/Cntr=0.3,0.1

Type RM Length L Ch R = 1 ,2560    ,69.4,68.7,68.1
XS GIS Cut Line= 2
2197158.06793418750706.7288453732197289.91858042750649.959817131
#Sta/Elev= 30
       0 1452.42     6.6 1450.81    15.4 1449.32    19.7 1448.33    24.1 1446.69
    28.4 1444.55    32.8 1442.83    37.1 1441.32    42.4 1439.63    45.8 1438.75
    54.5 1437.72    60.6 1435.82    63.7 1435.03    66.7 1434.48    69.8 1434.02
      72 1433.81    74.7 1434.17    76.3 1434.54    78.9 1435.38    80.7 1435.83
    81.9 1436.01    91.1 1436.64   106.3 1438.53   109.3 1439.08   111.2 1439.48
   115.2 1440.58   124.2 1444.17   128.6 1445.42   132.9  1446.5   143.6 1448.48
#Mann= 5 ,-1,0
       0      .1       0      30     .06       0    66.7    .045       0
    76.3     .06       0     140     .05       0
Bank Sta=66.7,76.3
XS Rating Curve= 0 ,0
Exp/Cntr(USF)=0,0
Exp/Cntr=0.3,0.1

Type RM Length L Ch R = 1 ,2491    ,68,71.9,75.3
XS GIS Cut Line= 4
2197177.60238794750761.3837473092197232.20993186750750.462238525
2197307.44699237750712.8437082712197341.42501969750688.573688751
#Sta/Elev= 30
       0 1448.43       3  1447.6    10.8 1444.99    14.9 1443.76      23  1442.3
    27.1 1441.65    31.2  1441.2    39.3 1439.81    47.5 1438.58    56.6 1436.87
    59.6  1436.2    64.6 1434.67    68.5 1433.68    71.5 1433.09    74.5 1432.71
    77.5 1433.03    82.5 1434.72    86.4 1435.33   101.3 1435.73   109.3 1436.22
   119.2 1437.45   127.2 1438.93   131.7 1440.04   136.1 1441.51     143 1444.12
   150.5 1447.17   159.9 1450.38   165.3 1451.53   175.1 1452.77   181.6 1454.28
#Mann= 5 ,-1,0
       0      .1       0      10     .06       0    71.5    .045       0
    77.5     .06       0  115.69     .05       0
Bank Sta=71.5,77.5
XS Rating Curve= 0 ,0
Exp/Cntr(USF)=0,0
Exp/Cntr=0.3,0.1

Type RM Length L Ch R = 1 ,2419    ,60.6,58.2,55.1
XS GIS Cut Line= 3
 2197188.5889171750831.2544557092197249.02046329750809.279348003
 2197328.3750189750805.006410393
#Sta/Elev= 30
       0 1446.97     3.8 1445.44     7.5 1444.08    16.6 1441.15    20.8 1440.07
    25.1 1439.16    29.4 1438.44    33.6 1437.96    42.1 1437.09    50.6 1436.46
    54.9 1436.35    59.1 1436.38    63.4 1436.61    67.5 1436.34    75.5 1434.18
    79.5 1433.69    83.5 1432.86    87.5 1432.77    91.5  1434.1    95.5 1434.79
    99.5  1434.8   103.5 1435.02   107.5 1435.63   111.5  1436.6   119.5 1438.96
   127.5 1441.46     131 1442.48   135.8 1443.51   139.6 1444.16   143.8 1444.74
#Mann= 4 ,-1,0
       0     .06       0    75.5    .045       0    91.5     .06       0
   104.3     .05       0
Bank Sta=75.5,91.5
XS Rating Curve= 0 ,0
Exp/Cntr(USF)=0,0
Exp/Cntr=0.3,0.1

Type RM Length L Ch R = 1 ,2361    ,48.5,47.3,45.8
XS GIS Cut Line= 3
2197205.07024788750887.4130642932197301.51655393750855.060822391
2197333.86879583750831.254455709
#Sta/Elev= 25
       0 1448.26     3.3 1447.17       7 1446.19    24.4 1441.99    35.8 1439.55
    41.2 1438.52    48.4 1437.54    53.9 1436.95    62.3 1436.45    66.6 1436.04
    70.8 1433.78   73.02 1432.69      75 1431.88    79.2 1432.48    79.81432.705
      80 1432.78    83.4  1434.1    87.7 1435.01    91.9 1435.47    95.1 1436.01
     110 1439.09     115 1439.87     125 1441.22   136.4 1443.02   141.9  1443.8
#Mann= 4 ,-1,0
       0     .06       0   73.02    .045       0    79.8     .06       0
      80     .05       0
Bank Sta=73.02,79.8
XS Rating Curve= 0 ,0
Exp/Cntr(USF)=0,0
Exp/Cntr=0.3,0.1

Type RM Length L Ch R = 1 ,2314    ,67.5,69.6,99.4
XS GIS Cut Line= 4
2197227.13372947750939.4419821152197253.57480053750927.833707016
2197318.06521775750894.9435942372197360.62889311750850.445206359
#Sta/Elev= 30
       0 1445.96     5.5 1444.91    14.2 1442.94    31.8  1439.5    41.7 1437.06
    45.3 1436.26    49.8 1435.62    54.2 1435.28    63.2 1435.19    65.5 1434.77
    67.7 1434.21    68.5 1433.91    71.4 1432.51    72.2 1432.21    74.4 1431.94
    76.7 1431.96    79.51432.506    85.7 1433.65    87.5 1433.84    94.7 1434.28
     104 1434.59   109.2 1434.87     121 1436.02   125.9 1437.03   135.1 1440.11
     139 1441.22   143.6 1442.35     148 1443.17   150.6 1443.55   162.8 1444.96
#Mann= 4 ,-1,0
       0     .06       0   68.88     .05       0    71.4    .045       0
    79.5     .05       0
Bank Sta=71.4,79.5
XS Rating Curve= 0 ,0
Exp/Cntr(USF)=0,0
Exp/Cntr=0.3,0.1

Type RM Length L Ch R = 1 ,2244    ,163.4,164.8,128.7
XS GIS Cut Line= 4
2197228.63807113751005.9129929252197305.25268678750973.990236403
2197362.71364852750955.4169962462197443.97157421750907.242654586
#Sta/Elev= 30
       0 1448.01     8.2 1445.12    16.8 1443.53    21.6 1443.01    25.5 1442.92
    29.8 1442.42    36.9 1441.16      43 1440.43    47.2 1439.65    60.2 1438.06
    86.1 1434.06    90.3  1433.3    94.5 1432.13    98.7 1431.59   102.9 1431.34
   107.1 1431.79   108.2 1432.11   111.3 1433.16   115.5 1434.02   143.4  1434.9
   175.3 1437.27     187 1438.34   192.8 1439.39   200.9 1441.73   207.4 1444.33
   210.5  1445.8   214.8 1447.48   218.4 1448.62   233.4 1451.81   237.9 1452.43
#Mann= 4 ,-1,0
       0     .06       0      60     .05       0    94.5    .045       0
   108.2     .05       0
Bank Sta=94.5,108.2
XS Rating Curve= 0 ,0
Exp/Cntr(USF)=0,0
Exp/Cntr=0.3,0.1

Type RM Length L Ch R = 1 ,2079    ,34.4,33.6,32.6
XS GIS Cut Line= 2
  2197245.968365751096.1765875042197501.12378226751010.717835312
#Sta/Elev= 30
       0 1444.18     4.1 1443.69    10.8 1442.31      22 1440.29    48.7 1436.22
    52.9 1435.82    61.4 1435.82    72.4 1434.49    78.3 1434.07    82.5 1433.95
    90.9 1434.04   107.8 1433.68   133.7 1434.31   141.5 1434.92   144.6 1434.94
     150  1434.6   158.4  1434.7   183.7  1434.5   187.9 1434.68   200.6 1435.99
   204.8  1435.4   208.1 1433.75   209.5 1433.14   212.7 1432.92   215.8 1433.63
   217.5 1433.98   225.9 1434.72   251.2 1437.57   256.9 1438.76   269.1  1442.3
#Mann= 5 ,-1,0
       0     .06       0      40     .07       0     170     .05       0
   208.1    .045       0   215.8     .05       0
#XS Ineff= 1 ,-1
   144.2  200.09 1436.57
Permanent Ineff=
       F
Bank Sta=208.1,215.8
XS Rating Curve= 0 ,0
Exp/Cntr(USF)=0,0
Exp/Cntr=0.3,0.1

Type RM Length L Ch R = 1 ,2046    ,110.4,25.3,25.3
XS GIS Cut Line= 5
2197263.22699102751164.7116929682197356.67613654 751111.31218124
2197439.00038379751068.5925718582197465.25514372751057.022677651
2197494.17987924751040.557828201
#Sta/Elev= 30
       0 1440.62     9.1 1439.49    23.2 1437.15    33.3 1435.92    44.3 1434.84
    47.3 1434.71    51.8  1435.1    56.4 1435.31      61 1434.73    65.6 1434.35
    79.4 1433.72   114.8 1433.26   123.7 1433.53   126.6 1433.73   129.6 1434.12
   143.1 1433.31   161.1 1433.04   170.2  1433.1   183.7 1433.48   195.1 1433.99
   209.9  1434.1   214.91433.888  216.66 1433.63   219.1 1433.21   222.1 1433.64
   223.5 1433.95   227.9 1434.95   228.7 1435.03   242.8 1436.05   262.4 1437.81
#Mann= 5 ,-1,0
       0      .1       0      50     .07       0   214.9    .045       0
   223.5     .07       0  249.07     .05       0
Bank Sta=216.66,222.1
XS Rating Curve= 0 ,0
Exp/Cntr(USF)=0,0
Exp/Cntr=0.3,0.1

Type RM Length L Ch R = 1 ,2021    ,27.9,120,122.9
XS GIS Cut Line= 6
2197277.24436285751180.0640525892197370.69350837751126.664540862
2197453.01775562 751083.944931482197471.70758472 751083.94493148
2197478.82751962751075.0450128592197508.19725107751055.910187823
#Sta/Elev= 30
       0 1438.98    10.1  1437.9    27.7 1435.25    42.4 1433.86    65.8 1432.76
    80.5 1432.46    86.4 1432.49   100.1 1432.13   109.3 1431.05   112.8 1431.29
   118.7 1431.97   128.2 1432.24   133.6 1432.11   142.5 1432.25   145.6 1432.45
   148.4 1432.36   154.3 1432.57   157.3 1432.44   180.3    1433   185.9 1432.96
   200.4 1433.43   203.5 1433.36   207.5 1432.98  209.83  1432.7   211.5  1432.5
   215.5 1432.54   216.71432.706   218.3 1433.03   250.1 1436.07   265.5 1438.37
#Mann= 5 ,-1,0
       0      .1       0      80     .07       0   207.5    .045       0
   218.3     .07       0  229.07     .05       0
Bank Sta=209.83,216.7
XS Rating Curve= 0 ,0
Exp/Cntr(USF)=0,0
Exp/Cntr=0.3,0.1

Type RM Length L Ch R = 1 ,1901    ,140.5,140,139.6
XS GIS Cut Line= 4
2197275.59503483751186.1892689892197339.17068846751152.195237161
2197413.28912723751149.9895202642197505.45879536751161.134006712
#Sta/Elev= 30
       0 1438.99     5.2 1438.38    14.3 1437.76    18.8 1437.16    24.8 1435.74
    30.7 1434.66    45.5 1432.94    61.5 1431.95    72.1 1431.54    77.1 1431.14
    85.1 1430.86   101.1 1430.72   105.1 1430.52   109.1 1429.85   113.1 1429.24
   115.4 1429.76   117.1 1430.15   121.1  1430.8   129.1 1430.86   146.2 1431.28
   193.5  1431.6   197.5 1431.81   201.5 1432.46   205.6  1433.6   209.6 1435.01
   219.2 1438.82   221.7 1439.72   225.7 1440.87   229.7  1441.7   239.1  1442.9
#Mann= 4 ,-1,0
       0      .1       0   109.1    .045       0   115.4     .07       0
  216.24     .05       0
Bank Sta=109.1,115.4
XS Rating Curve= 0 ,0
Exp/Cntr(USF)=0,0
Exp/Cntr=0.3,0.1

Type RM Length L Ch R = 1 ,1761    ,52,48,42.3
XS GIS Cut Line= 2
2197285.61701063751298.1192451432197467.28651593751283.608901269
#Sta/Elev= 28
       0 1435.61     2.6 1435.55     6.6 1435.25    10.6 1434.19    14.6 1432.53
    18.1 1431.76    26.6 1430.52    30.7 1430.12    34.7 1429.92    50.7 1429.59
    58.7 1429.31    70.1  1429.4    82.8 1429.39    86.8 1429.23    92.4 1428.45
    94.9 1428.02    98.9 1428.18     1011428.481   102.9 1428.76   110.9 1429.25
     135 1429.58     147 1429.97   159.1  1430.6   163.1 1431.06   167.1 1431.95
   175.1 1434.18   179.1 1435.12   182.2 1435.72
#Mann= 3 ,-1,0
       0     .05       0    92.4    .045       0     101     .07       0
Bank Sta=92.4,101
XS Rating Curve= 0 ,0
Exp/Cntr(USF)=0,0
Exp/Cntr=0.3,0.1

Type RM Length L Ch R = 1 ,1713    ,32.1,32.2,33.2
XS GIS Cut Line= 4
2197337.31492001751369.6422749232197350.57489669751357.389124427
2197419.07754726751319.407456786 2197484.1889775 751276.67808069
#Sta/Elev= 26
       0 1431.24    22.3 1430.44    26.7 1430.16      29 1429.86      37  1429.2
    43.2  1428.5    48.8  1428.3    51.5 1427.99    54.7 1427.86    56.5 1427.64
    59.7  1427.6      61 1427.64   62.27 1427.84    63.5  1428.1    69.4 1428.85
    74.8 1429.24    88.5 1429.67   110.3 1430.84   130.6 1431.53   133.4 1431.75
   136.3 1432.05   139.2 1432.53   150.3 1434.76   159.4 1436.27   166.1 1437.11
   174.3 1437.91
#Mann= 4 ,-1,0
       0     .05       0    54.7    .045       0   62.27     .07       0
  166.38     .05       0
Bank Sta=54.7,62.27
XS Rating Curve= 0 ,0
Exp/Cntr(USF)=0,0
Exp/Cntr=0.3,0.1

Type RM Length L Ch R = 1 ,1680    ,25.2,27.4,30.5
XS GIS Cut Line= 4
2197346.92683212751401.2814856212197369.87260204751381.489659125
2197438.37525261751343.5079914842197503.48668285751300.778615388
#Sta/Elev= 26
       0 1429.35    12.2 1429.12    30.3 1429.16    37.5 1428.95    42.1 1428.65
      44  1428.3    46.7 1427.63    49.7 1426.61    51.2  1426.1    52.8 1425.96
    55.8 1425.88    58.7  1426.6      65 1428.34    69.5 1428.98    74.1 1429.25
    87.8 1429.55    92.4 1429.75   110.8 1430.93   117.4 1431.49   120.4 1431.66
   128.9 1432.49   134.7 1432.94   154.9 1434.06   166.5 1435.21     173 1435.97
   186.5 1437.29
#Mann= 4 ,-1,0
       0     .05       0    49.7    .045       0    58.7     .07       0
  158.63     .05       0
Bank Sta=49.7,58.7
XS Rating Curve= 0 ,0
Exp/Cntr(USF)=0,0
Exp/Cntr=0.3,0.1

Type RM Length L Ch R = 1 ,1653    ,10.5,10.3,10.3
XS GIS Cut Line= 2
2197342.12087607751409.691908718 2197492.5120292751374.002977315
#Sta/Elev= 26
       0 1429.59     6.2 1428.99    14.4 1428.61    26.8 1428.46      35  1428.5
    43.2  1428.3    47.3 1427.96    48.6 1427.76    53.61426.682    55.6 1426.22
    58.6 1426.47    59.7 1426.64    63.8 1427.57    67.9 1428.01    71.5 1428.26
    76.1 1428.52    88.5 1428.81   106.2 1429.38     109 1429.49   111.8 1429.75
   117.2 1430.45   125.4  1431.8   133.7 1432.66   137.8 1433.16   141.9  1433.8
   154.6 1436.48
#Mann= 5 ,-1,0
       0     .05       0      40     .07       0    53.6    .045       0
    59.7     .07       0     140     .05       0
Bank Sta=53.6,59.7
XS Rating Curve= 0 ,0
Exp/Cntr(USF)=0,0
Exp/Cntr=0.3,0.1

Type RM Length L Ch R = 1 ,1643    ,15.3,15.7,16.5
XS GIS Cut Line= 2
2197319.87917097751425.2946489192197490.11843128751385.278249083
#Sta/Elev= 26
       0 1433.34     4.4  1432.6       7 1431.84    12.6 1430.37    16.7 1429.79
    29.1 1428.76    33.2 1428.58    45.5 1428.29      66 1428.34    70.2 1428.16
    74.3 1427.56    78.4 1426.58    82.5 1426.07    85.61426.562    86.6 1426.71
    90.7 1427.61    94.8 1427.99    98.9 1428.22     103  1428.4   131.8 1429.13
   139.9 1429.49   143.4  1429.8   160.6 1431.96   164.7 1432.54   168.8 1433.25
   174.9 1434.58
#Mann= 5 ,-1,0
       0     .05       0      70     .07       0    78.4    .045       0
    85.6     .07       0     170     .05       0
Bank Sta=78.4,85.6
XS Rating Curve= 0 ,0
Exp/Cntr(USF)=0,0
Exp/Cntr=0.3,0.1

Type RM Length L Ch R = 1 ,1627    ,40,39.4,38.1
XS GIS Cut Line= 3
2197326.06448554751446.1423454282197389.14118359751424.438535348
2197502.40794244751398.665260877
#Sta/Elev= 28
       0 1433.33       3 1432.92     5.6  1432.3     6.5 1431.98    10.7  1430.9
    14.9 1429.98    19.2 1429.55    27.5    1429    30.7 1428.96    39.8 1428.51
    43.3 1428.42    48.8  1428.4    61.5 1428.64    65.4 1428.58    69.8 1428.23
      72 1427.81    76.81426.651      78 1426.35      82 1426.04    86.2 1426.55
    94.4 1427.92   106.7 1428.28   143.7 1428.92   147.8 1429.06   155.5 1429.53
   160.1 1429.92   164.2 1430.43   182.9 1433.61
#Mann= 6 ,-1,0
       0     .07       0      30     .05       0      60     .07       0
    76.8    .045       0    86.2     .07       0  166.71     .05       0
Bank Sta=76.8,86.2
XS Rating Curve= 0 ,0
Exp/Cntr(USF)=0,0
Exp/Cntr=0.3,0.1

Type RM Length L Ch R = 1 ,1588    ,46.5,45.7,44.7
XS GIS Cut Line= 3
2197341.66409904751477.3415724192197404.74079708751455.637762338
2197518.00755594751429.864487868
#Sta/Elev= 30
       0 1433.73     6.9 1433.98    15.3 1434.58    40.7 1434.79    49.7 1435.09
    53.4 1435.07    61.9 1433.94    70.2 1433.27    74.3 1432.67    78.4 1431.09
    82.5 1428.59    86.6 1426.49    89.7 1425.74    90.7  1425.5    94.8 1425.31
    98.21425.798    99.9 1426.34     103 1427.67     105  1428.3   107.1 1428.88
   108.4 1428.98   111.3 1429.11     140 1429.32   156.4    1429   160.5 1428.99
   164.6 1429.14   168.7 1430.02   172.8 1432.15   176.9 1433.94   182.9 1436.04
#Mann= 5 ,-1,0
       0     .07       0      40     .08       0    89.7    .045       0
    98.2     .08       0  146.71     .05       0
Bank Sta=89.7,98.2
XS Rating Curve= 0 ,0
Exp/Cntr(USF)=0,0
Exp/Cntr=0.3,0.1

Type RM Length L Ch R = 1 ,1542    ,70.5,70.5,70.3
XS GIS Cut Line= 3
 2197340.8211696751525.8507993392197499.73829647751474.789250893
 2197548.3936181751469.481397624
#Sta/Elev= 30
       0 1433.72     3.5 1433.53     7.7 1433.54    28.7 1434.66    66.5 1434.81
    74.9 1434.67    91.8 1433.84      96 1433.28    98.6 1432.37   100.2 1431.76
   104.4 1429.12   108.1 1427.28   112.8 1426.12     117 1425.14   120.9  1426.1
   125.4 1427.69   129.6 1428.14     138 1428.44   142.2 1428.75   150.6 1429.65
   158.9 1430.81   163.2 1431.06   167.4 1431.62   171.4 1433.37   175.4 1435.86
   179.4 1437.46   187.5 1440.02   199.5 1444.53   203.6 1445.66   215.9 1447.87
#Mann= 5 ,-1,0
       0     .07       0      50     .08       0   112.8    .045       0
   120.9     .08       0     150     .05       0
Bank Sta=112.8,120.9
XS Rating Curve= 0 ,0
Exp/Cntr(USF)=0,0
Exp/Cntr=0.3,0.1

Type RM Length L Ch R = 1 ,1471    ,79.9,80.7,81.6
XS GIS Cut Line= 4
2197377.43188033751584.2184483172197432.33547048751570.891642941
2197504.41742845751546.8643236172197561.20927412751540.311418347
#Sta/Elev= 29
       0 1433.66    27.5 1433.97    77.4 1433.62    81.6 1433.38      83 1433.04
    86.2 1432.07    90.1 1430.23    94.3  1427.9    95.7 1427.2698.458891426.157
     102 1425.18   102.7 1425.07   105.2  1425.5106.95891426.032   111.1 1428.15
   114.6 1429.17   124.1 1431.44   132.5 1433.35   140.3 1435.49   144.3 1437.22
   148.3  1439.1   152.4 1440.63   160.4 1443.86   168.5 1447.64   172.5 1448.69
   176.5 1449.55   180.6 1450.28   184.6 1450.87   189.6 1451.81
#Mann= 4 ,-1,0
       0     .05       0      10     .08       098.45889    .045       0
106.9589     .03       0
Bank Sta=98.45889,106.9589
XS Rating Curve= 0 ,0
Exp/Cntr(USF)=0,0
Exp/Cntr=0.3,0.1

Type RM Length L Ch R = 1 ,1391    ,50.6,51.4,52.3
XS GIS Cut Line= 3
2197404.99857505751653.1351850962197438.88837575751647.342204424
2197557.93282149751620.038432466
#Sta/Elev= 25
       0 1434.32    23.5 1433.72    52.1 1433.44    68.5 1433.19    72.6 1432.73
    76.7 1431.44    80.8 1429.72      84 1428.06    84.9 1427.52    89.1 1425.82
90.218571425.536    93.2 1424.78    97.3 1424.8198.318581425.436   101.4 1427.34
   105.5 1429.65   120.7 1435.48   121.9 1435.91     126 1437.11   134.2 1439.85
   138.3 1441.06   146.5 1445.04   150.6 1446.31   154.7 1447.06   156.5 1447.27
#Mann= 5 ,-1,0
       0     .07       0   74.38     .05       090.21857    .045       0
98.31858     .05       0  104.38     .03       0
Bank Sta=90.21857,98.31858
XS Rating Curve= 0 ,0
Exp/Cntr(USF)=0,0
Exp/Cntr=0.3,0.1

Type RM Length L Ch R = 1 ,1339    ,55.2,57,59.3
XS GIS Cut Line= 3
2197433.45565966751694.4874137352197533.77408644  751680.9523879
2197571.99062998751648.309090296
#Sta/Elev= 28
       0 1432.97    18.9 1433.08    22.9 1433.01    43.1 1432.38    51.2 1431.92
    55.2 1430.94    59.3 1429.39    63.3 1427.41    67.61425.632    71.4 1424.06
    75.4 1424.67      771425.578    79.4 1426.94    83.5 1428.36    87.5 1429.56
    95.6 1431.68    99.5 1432.52   114.9 1436.25   119.4 1437.53   122.6 1438.79
   125.4 1440.08   128.3  1441.7   130.7 1443.14     134 1444.48   135.9 1445.16
   137.8 1445.48   146.5 1446.54   151.5 1447.45
#Mann= 4 ,-1,0
       0     .07       0      50     .05       0    67.6    .045       0
      77     .05       0
Bank Sta=67.6,77
XS Rating Curve= 0 ,0
Exp/Cntr(USF)=0,0
Exp/Cntr=0.3,0.1

Type RM Length L Ch R = 1 ,1282    ,72.3,71.4,70.4
XS GIS Cut Line= 3
2197440.62126158751734.2963132512197549.69764625751745.442805116
2197603.83774959751760.570186932
#Sta/Elev= 29
       0 1432.63    11.6 1432.37    23.1  1432.3    31.7 1432.12    38.7  1431.6
    47.8 1430.77    51.8  1430.3    55.8 1429.17    63.9 1425.67    67.31424.327
    67.9 1424.09    71.9 1423.57    74.61424.298    75.9 1424.68      80 1425.45
      84 1425.56      88 1426.03      92 1426.86    96.1  1427.9   100.1 1429.18
   112.2 1433.67   128.8 1439.21   134.2 1440.86   141.3 1443.18   145.4 1444.44
   153.6 1446.49   157.9 1447.75   162.1 1449.24   165.9 1450.39
#Mann= 5 ,-1,0
       0      .1       0      40     .07       0    67.3    .045       0
    74.6     .07       0  139.64     .05       0
Bank Sta=67.3,74.6
XS Rating Curve= 0 ,0
Exp/Cntr(USF)=0,0
Exp/Cntr=0.3,0.1

Type RM Length L Ch R = 1 ,1211    ,45.3,45.8,46
XS GIS Cut Line= 3
2197382.65612635751814.4248847022197544.52707355751811.200363842
2197594.18469481751801.526801259
#Sta/Elev= 30
       0 1435.49     5.5 1435.28     9.5 1434.81    13.5  1434.5    21.5 1434.25
    33.5 1433.47    53.5 1432.97    69.5 1432.34    81.5  1431.5    93.5 1430.87
    97.5 1430.52   105.5 1429.42   109.5 1427.96   113.5 1426.13   117.5  1424.1
   118.21423.907   121.5    1423   124.3  1423.9   125.5 1424.32   129.5 1424.76
   137.5 1424.54   141.5 1424.61   145.5 1425.16   149.5  1426.5   157.6 1429.91
   170.1 1435.68   177.8 1438.84     186 1441.67   190.1 1442.96   212.5 1449.56
#Mann= 5 ,-1,0
       0      .1       0     100     .07       0   118.2    .045       0
   124.3     .07       0   201.9     .05       0
Bank Sta=118.2,124.3
XS Rating Curve= 0 ,0
Exp/Cntr(USF)=0,0
Exp/Cntr=0.3,0.1

Type RM Length L Ch R = 1 ,1165    ,88.7,88.5,88.5
XS GIS Cut Line= 2
2197415.59270212751856.480004762 2197588.5449387751857.158248827
#Sta/Elev= 30
       0 1433.84    12.6 1433.26    20.6 1433.02    32.6 1432.22    40.6 1432.01
    48.6 1431.64    56.6 1431.47    64.6  1431.1    68.6 1430.42    72.6 1428.51
    80.6 1423.68    84.6 1423.13   86.47 1423.67    88.6 1424.22    92.6 1424.56
   100.6 1424.25   104.6 1424.19   108.6 1424.22   112.6 1424.38   116.6 1424.78
   120.6 1425.69   124.6 1427.07   128.8 1428.78   132.8 1430.56   140.4 1434.25
   144.5 1436.13   148.6 1437.88   152.6 1439.38   160.6 1442.04     173 1446.86
#Mann= 5 ,-1,0
       0      .1       0      70     .07       0    80.6    .045       0
   86.47     .07       0     170     .05       0
Bank Sta=80.6,86.47
XS Rating Curve= 0 ,0
Exp/Cntr(USF)=0,0
Exp/Cntr=0.3,0.1

Type RM Length L Ch R = 1 ,1077    ,73.2,73.5,73.5
XS GIS Cut Line= 2
2197434.58353594751944.6517332132197623.13538602751944.651733213
#Sta/Elev= 30
       0 1432.34     5.6 1432.07    13.6 1431.85    21.6  1431.5    33.6 1431.27
    45.6 1430.85    49.6 1430.24    53.6 1428.31    57.6 1425.46    60.91423.249
    61.6 1422.78    65.6 1422.54    67.51423.058    69.6 1423.63    73.6 1423.88
    81.6 1423.54    89.6 1423.41   105.6 1423.41   117.6 1423.54   133.6  1424.2
   141.6 1424.71   145.1 1425.08   149.6 1425.72   153.6 1426.55   157.6 1427.74
   165.6 1430.79   169.6 1432.14   173.6 1433.32   185.6 1436.24   188.6 1436.87
#Mann= 5 ,-1,0
       0      .1       0      50     .07       0    60.9    .045       0
    67.5     .07       0     150     .05       0
Bank Sta=60.9,67.5
XS Rating Curve= 0 ,0
Exp/Cntr(USF)=0,0
Exp/Cntr=0.3,0.1

Type RM Length L Ch R = 1 ,1003    ,84.9,84.9,84.4
XS GIS Cut Line= 2
2197442.72246472 752017.223848172197628.56133854  752018.5803363
#Sta/Elev= 28
       0 1431.84     5.5 1431.69    13.5 1431.75    25.5 1431.69    29.5 1431.52
    33.2 1430.87    33.5 1430.81    37.5 1429.13    41.5 1426.41    45.8 1424.03
    49.5 1422.38      511422.069    53.5 1421.55    55.91422.137    57.9 1422.55
    61.5 1422.83    69.5 1422.64    81.5 1423.05   102.2 1423.28   121.5 1423.71
   133.5  1424.2   149.5 1425.13   157.5 1425.98   161.5 1426.66   169.5 1428.19
   173.5  1429.2   181.5 1431.43   185.8 1432.43
#Mann= 5 ,-1,0
       0      .1       0      40     .07       0      51    .045       0
    55.9     .07       0     140     .05       0
Bank Sta=51,55.9
XS Rating Curve= 0 ,0
Exp/Cntr(USF)=0,0
Exp/Cntr=0.3,0.1

Type RM Length L Ch R = 1 ,918     ,36.9,36.9,36.9
XS GIS Cut Line= 2
2197446.79192911752102.0043562972197606.17928439752097.256647842
#Sta/Elev= 26
       0  1430.9     2.1 1430.74     9.4 1430.44    17.4 1430.39    21.4 1430.09
    25.4 1429.16    33.4 1424.84    37.4 1423.24      431421.618    45.4 1420.89
    49.4 1421.37    50.31421.613    53.4 1422.45    57.4 1422.69    61.4 1422.54
    69.4 1422.65    77.4 1422.91    93.4 1423.23   101.4 1423.51   113.4 1423.64
   125.4  1424.2   137.4 1424.89   149.4 1425.79   153.5 1426.19   157.5 1426.84
   159.5 1427.24
#Mann= 5 ,-1,0
       0      .1       0      40     .06       0      43    .045       0
    50.3     .06       0     130      .1       0
Bank Sta=43,50.3
XS Rating Curve= 0 ,0
Exp/Cntr(USF)=0,0
Exp/Cntr=0.3,0.1

Type RM Length L Ch R = 1 ,881     ,38.7,37.1,34.9
XS GIS Cut Line= 3
2197446.91011787752138.8546661112197571.43572821 752135.19214816
2197678.86958811752100.398227625
#Sta/Elev= 30
       0 1432.59     5.3 1431.14     9.3 1430.83    13.3 1430.77    17.3 1430.47
    21.3 1429.75    25.3 1428.23    33.3 1424.38    37.3    1423    41.3  1421.8
    45.3 1420.84    49.3 1420.91    53.2 1421.63    57.3 1422.16    61.3 1422.38
    73.3 1422.59    89.3 1423.17   105.3 1423.92   125.4 1425.32   129.6 1425.68
   133.8 1426.24   146.4 1426.88   152.2 1427.28   164.9 1428.62     180 1430.63
   188.4 1431.35     209    1434   217.9 1435.25   230.5 1437.61   237.5 1438.63
#Mann= 5 ,-1,0
       0      .1       0      40     .07       0    41.3    .045       0
    53.2     .07       0  134.58      .1       0
Bank Sta=41.3,53.2
XS Rating Curve= 0 ,0
Exp/Cntr(USF)=0,0
Exp/Cntr=0.3,0.1

Type RM Length L Ch R = 1 ,844     ,39.2,39.3,39.3
XS GIS Cut Line= 3
2197443.24759992752181.5840422072197538.47306665752162.050613135
2197676.42790947752120.542076356
#Sta/Elev= 30
       0 1433.63       5 1433.62    21.4 1432.62    25.4 1432.25    29.5  1430.6
    37.7    1422    39.71421.297    41.8 1420.63    45.9 1420.59    49.9 1421.14
      54 1421.95    58.7 1422.55    70.4 1423.06    82.9 1423.75    97.2 1424.73
   115.7 1425.46   119.9 1425.85     125 1426.11   132.4 1426.77   136.6 1427.04
   144.9 1427.42   153.3 1427.63   161.6 1427.62   174.2 1427.88   182.8 1428.31
   189.2 1428.89   214.9 1431.75   224.5 1433.08   230.9 1433.75   241.3 1435.08
#Mann= 4 ,-1,0
       0      .1       0    39.7    .045       0    49.9     .07       0
  137.21      .1       0
Bank Sta=39.7,49.9
XS Rating Curve= 0 ,0
Exp/Cntr(USF)=0,0
Exp/Cntr=0.3,0.1

Type RM Length L Ch R = 1 ,805     ,25.4,24.3,23.5
XS GIS Cut Line= 3
2197444.46843924752221.2613200112197539.69390596752201.727890938
2197677.64874879752160.219354159
#Sta/Elev= 30
       0 1432.75     7.9 1432.87      12 1432.23      16 1430.46    20.3 1428.21
    28.3 1424.38    32.4 1423.23    36.4 1422.63    40.6 1422.29    43.9 1422.17
    47.41421.461    48.7 1421.09    52.8  1420.8      56 1421.37    60.9 1422.21
      65  1422.4    93.6 1422.96    97.2 1422.93   106.1  1423.5   117.3 1423.83
   122.8 1423.82   131.1 1424.26     152 1424.99   160.4 1425.43   177.1 1425.58
   189.6  1426.4   200.8 1427.85   227.2 1429.16   231.4 1429.56   241.3 1431.17
#Mann= 6 ,-1,0
       0      .1       0      40     .07       0    47.4    .045       0
      56     .07       0  137.21      .1       0  241.27     .07       0
Bank Sta=47.4,56
XS Rating Curve= 0 ,0
Exp/Cntr(USF)=0,0
Exp/Cntr=0.3,0.1

Type RM Length L Ch R = 1 ,781     ,56,58.5,57.3
XS GIS Cut Line= 2
2197453.01431446752248.119784985 2197649.5694445752191.350756743
#Sta/Elev= 29
       0 1432.31     3.3 1432.36     7.5 1431.92    11.4 1430.54    19.9 1425.74
    24.1 1423.68    27.5 1422.29    28.3 1422.04    32.4 1421.66    40.8 1421.84
    44.9 1421.77    49.1 1421.35   51.02 1420.99    53.3 1420.56    57.4 1420.75
    58.6 1420.99    61.6 1421.59    65.7 1421.92    82.5 1421.91      94  1422.1
   103.2 1422.63   111.5 1422.91   130.9 1423.08   154.8 1423.41   186.5  1423.6
   190.6 1423.98   194.8  1424.8   203.1 1427.18   204.6 1427.55
#Mann= 5 ,-1,0
       0      .1       0      30     .07       0   51.02    .045       0
    58.6     .07       0     130      .1       0
Bank Sta=51.02,58.6
XS Rating Curve= 0 ,0
Exp/Cntr(USF)=0,0
Exp/Cntr=0.3,0.1

Type RM Length L Ch R = 1 ,722     ,38.8,36.2,29.3
XS GIS Cut Line= 3
2197449.96221616752302.4471345932197644.07566757752247.509365327
2197724.65106249752243.846847376
#Sta/Elev= 30
       0 1430.83    10.6 1431.38    14.8 1431.24    18.9    1430    23.1 1428.12
    27.2 1425.97    31.4 1424.34    35.6 1423.25    39.7 1422.55    54.7 1421.21
    57.9 1420.66    60.5 1420.02   65.41 1420.69    68.8 1421.49      73 1421.65
    85.4 1421.48    97.9 1421.93   110.4 1421.87   168.6 1422.44   181.1 1423.16
   217.9 1425.74   221.9 1426.45   225.9 1427.78   229.9 1428.72   234.7 1429.47
   238.5 1429.88   257.9 1430.81   261.9 1431.21   273.9 1433.07   282.4 1433.91
#Mann= 5 ,-1,0
       0      .1       0      30     .07       0    57.9    .045       0
   65.41     .07       0     140      .1       0
Bank Sta=57.9,65.41
XS Rating Curve= 0 ,0
Exp/Cntr(USF)=0,0
Exp/Cntr=0.3,0.1

Type RM Length L Ch R = 1 ,686     ,37.7,39.1,43.3
XS GIS Cut Line= 6
2197448.81469047752341.849579341 2197481.3778486752334.406571769
2197534.40927755752302.773789588 2197589.3014584752282.305518764
2197640.41314962752272.5365713262197729.67025465752266.282677251
#Sta/Elev= 30
       0 1429.72    11.7 1430.42    15.8  1430.5    19.9  1430.4      24 1429.51
    32.2 1426.74    35.8 1425.81    45.1 1424.32      48 1423.27    51.4 1421.58
    53.8 1420.94    56.8 1420.42    59.2 1420.08    64.6 1419.73    69.81420.443
    78.6  1421.6    83.2 1421.73    97.8 1421.78   105.6 1421.63   126.9  1421.7
   148.3 1422.13   181.1 1422.47   205.8 1423.66   221.6 1424.94   233.6 1426.29
   245.6 1428.11   253.8 1429.11   269.7 1430.71   285.7 1432.01   295.2 1433.23
#Mann= 5 ,-1,0
       0      .1       0      30     .06       0    56.8    .045       0
    69.8     .07       0  145.15      .1       0
Bank Sta=56.8,69.8
XS Rating Curve= 0 ,0
Exp/Cntr(USF)=0,0
Exp/Cntr=0.3,0.1

Type RM Length L Ch R = 1 ,647     ,23.4,23.8,24.4
XS GIS Cut Line= 6
2197461.22953406752376.7681702532197493.79269219752369.325162681
2197532.97928972752347.6181893232197546.21370149752326.094406988
2197601.71630199752305.0157165062197734.76006234752288.382455334
#Sta/Elev= 30
       0 1429.65    11.2  1429.6    23.5 1430.03    33.4 1429.41    40.7 1427.61
      47 1425.47    49.8 1424.41    55.9 1421.35      59 1419.95    63.6  1419.6
    68.1  1421.3      75 1424.98    79.4 1426.41    90.5 1427.08    96.8 1427.04
   103.5  1426.5   108.8 1427.69   111.9 1427.94   130.5 1427.87   139.8 1427.04
   161.2 1426.07   169.5 1426.47   180.4  1425.9   188.2 1426.31   198.8 1425.95
   217.2 1426.53   235.5 1427.55   267.1 1431.62   287.1 1435.67   297.6 1437.35
#Mann= 6 ,-1,0
       0      .1       0      20     .06       0    55.9    .045       0
    68.1     .06       0  113.47     .07       0  143.47      .1       0
Bank Sta=55.9,68.1
XS Rating Curve= 0 ,0
Exp/Cntr(USF)=0,0
Exp/Cntr=0.3,0.1

Type RM Length L Ch R = 1 ,623     ,71.1,70.5,69.9
XS GIS Cut Line= 4
2197464.00186831752378.7495919072197503.06872645752389.126726102
 2197574.4878265752355.553644883 2197739.3011343752318.928465373
#Sta/Elev= 30
       0 1429.66     8.5 1429.68    16.7 1430.42    20.9 1430.56    29.1 1430.41
    37.4 1429.86    41.6 1429.24    49.7    1427    54.9 1424.77    63.7 1421.68
    68.2 1420.37    71.3 1420.13    72.6 1420.23    76.2  1421.6    89.3 1428.43
   103.5 1435.23   107.9 1436.82   119.3 1440.46   125.2 1441.86   129.3 1442.61
   157.9 1445.98   178.4 1448.89   218.5 1452.08   223.3 1452.11   231.7 1451.45
     244 1451.46   256.3 1452.19   266.9 1452.47   280.9 1453.15   288.2 1453.19
#Mann= 7 ,-1,0
       0      .1       0      20     .06       0    63.7    .045       0
    76.2     .06       0  129.34     .07       0  229.34     .06       0
  279.34      .1       0
Bank Sta=63.7,76.2
XS Rating Curve= 0 ,0
Exp/Cntr(USF)=0,0
Exp/Cntr=0.3,0.1

Type RM Length L Ch R = 1 ,553     ,14.3,22.1,31.3
XS GIS Cut Line= 4
2197459.36878217752397.2364410772197552.40637682 752444.68561435
2197584.03915901752427.0084713662197775.69660399752415.843960007
#Sta/Elev= 30
       0 1429.22     9.9 1429.24    18.4 1429.65    27.8 1429.38    35.1 1428.64
    45.2 1427.13      66 1423.57    74.9 1422.32    83.8 1421.55   104.4 1420.94
   109.8 1420.42   113.9 1419.32  116.46 1418.11   118.6 1417.29   121.5 1417.19
   122.5  1417.3   124.5 1418.12   127.1 1419.33   131.7 1421.62   136.2 1422.87
   140.7 1423.02   144.8 1422.55   152.8  1421.1   155.9 1421.27   164.9 1422.41
     258 1424.88     277 1426.05   305.1 1428.99   321.1 1430.24   332.7 1431.48
#Mann= 6 ,-1,0
       0      .1       0      30     .06       0   113.9    .045       0
   127.1     .06       0  134.44     .07       0  240.68     .06       0
Bank Sta=116.46,124.5
XS Rating Curve= 0 ,0
Exp/Cntr(USF)=0,0
Exp/Cntr=0.3,0.1

Type RM Length L Ch R = 1 ,530     ,47.9,47.4,45.5
XS GIS Cut Line= 5
2197433.31825567752408.4009524352197555.19750466752453.989373815
2197604.50742983752462.3627573332197644.51359553752465.153885173
2197784.06998751752445.615990296
#Sta/Elev= 30
       0 1427.24    20.1 1428.62    33.9 1428.78    37.2  1428.7    41.5 1428.24
      50 1426.31    62.8 1424.33    75.7 1423.42      93 1421.85     105 1421.38
   122.6 1421.14   135.2 1420.52   139.2  1419.5   144.2 1417.59   147.3 1416.66
   151.4 1416.18   155.5 1416.12   159.5 1417.47   163.6 1419.75     165 1420.03
   167.6 1420.36   183.8 1421.38   207.9 1421.83     228 1421.81   256.3 1422.57
   276.4 1423.38   296.6  1425.2     312  1427.2   341.1 1430.48   361.2 1432.43
#Mann= 6 ,-1,0
       0      .1       0      50     .06       0   144.2    .045       0
   159.5     .06       0  160.13     .07       0  260.25     .05       0
Bank Sta=144.2,159.5
XS Rating Curve= 0 ,0
Exp/Cntr(USF)=0,0
Exp/Cntr=0.3,0.1

Type RM Length L Ch R = 1 ,483     ,30.2,28.6,27.1
XS GIS Cut Line= 5
2197429.13156391752449.802682055 2197551.0108129752495.391103435
2197600.32073807752503.7644869542197640.32690377752506.555614793
2197779.88329575752487.017719916
#Sta/Elev= 30
       0  1426.6    16.1 1427.62    28.9 1427.77      33 1427.19    41.7 1425.04
      46 1424.23    58.8 1423.41    67.3 1423.29    98.2 1420.96   131.3 1420.37
   151.6 1420.42   155.7 1420.03   159.7 1418.97   163.9 1416.94   167.8 1415.39
   171.9 1414.59   175.9 1415.12  176.45 1415.45     180 1417.58     184 1419.14
     188 1419.63     196 1419.85   236.2 1419.88   253.2 1420.76   268.6  1421.2
   276.6 1421.92   296.8 1424.87   313.4 1426.84   353.4 1429.09   361.2 1429.96
#Mann= 6 ,-1,0
       0      .1       0      60     .06       0  160.13     .07       0
   167.8    .045       0  176.45     .07       0  260.25     .05       0
Bank Sta=167.8,176.45
XS Rating Curve= 0 ,0
Exp/Cntr(USF)=0,0
Exp/Cntr=0.3,0.1

Type RM Length L Ch R = 1 ,454     ,86,85.4,84.3
XS GIS Cut Line= 4
2197424.94487215752492.1347876222197533.79885789752529.349825483
2197656.60848283752532.1409533232197777.55735588752507.951178713
#Sta/Elev= 30
       0 1426.12    11.9  1426.7    20.3 1426.84    24.6 1426.35    37.2 1422.78
    41.5 1422.17    71.1 1420.66   102.1 1419.94   121.7 1419.17   137.4  1419.2
   149.4 1419.49   153.4  1419.3   157.4 1417.68   161.4 1414.73   165.4 1412.86
   169.4  1412.5   173.4 1413.03   177.4 1414.79   181.4 1417.75   185.4 1419.28
   201.4 1419.69   225.4 1419.59   232.3 1419.38   237.4  1418.9   249.7 1420.05
   270.1 1420.81   286.4 1422.77     319 1425.87   355.7    1428   361.2 1428.58
#Mann= 6 ,-1,0
       0      .1       0      60     .06       0      90     .07       0
   161.4    .045       0   177.4     .07       0  257.88     .05       0
Bank Sta=161.4,177.4
XS Rating Curve= 0 ,0
Exp/Cntr(USF)=0,0
Exp/Cntr=0.3,0.1

Type RM Length L Ch R = 1 ,369     ,22.7,23,23.2
XS GIS Cut Line= 2
2197515.26536527752620.1012348092197704.25129154752608.564303263
#Sta/Elev= 28
       0 1419.43     4.9 1419.15    20.9 1418.86      33 1418.91      49 1418.53
      61  1418.1      65 1417.79      69 1417.26      73 1415.83    76.2 1413.98
    77.1 1413.46    81.1 1412.02    85.1 1412.51    86.11413.141    86.7 1413.52
    89.1 1414.95    93.1 1417.54    97.1 1418.46   101.1 1418.72   109.1    1419
   117.1 1419.07   129.1  1418.9   141.2 1418.95   153.2 1419.23   165.2 1419.09
   168.6 1419.12   177.2 1419.22   189.3  1419.7
#Mann= 4 ,-1,0
       0     .07       0    76.2    .045       0    86.1     .07       0
     160     .05       0
Bank Sta=77.1,86.7
XS Rating Curve= 0 ,0
Exp/Cntr(USF)=0,0
Exp/Cntr=0.3,0.1

Type RM Length L Ch R = 1 ,346     ,63.1,63,63
XS GIS Cut Line= 2
2197508.12345526752641.526964823   2197706.99818752633.835677125
#Sta/Elev= 29
       0 1419.84     8.1 1419.19    37.2 1418.91    44.1 1418.72    48.1 1418.53
    60.1 1418.38    68.1 1418.09    72.1 1417.86    76.1 1417.35    80.1 1415.94
      841413.678   85.12 1413.23    88.1 1412.07    92.1 1413.23    93.91414.413
    96.1 1415.86   100.1 1417.52   104.1 1418.22     108 1418.49   116.1 1418.81
   136.2  1418.6   144.2 1418.62   148.2 1418.43   152.2 1418.52   156.2 1418.75
   172.2  1418.8   180.2  1418.9   188.2 1419.11     199  1419.6
#Mann= 5 ,-1,0
       0     .07       0      70     .06       0      84    .045       0
    93.9     .06       0     170     .05       0
Bank Sta=85.12,92.1
XS Rating Curve= 0 ,0
Exp/Cntr(USF)=0,0
Exp/Cntr=0.3,0.1

Type RM Length L Ch R = 1 ,283     ,33.8,33.7,33.6
XS GIS Cut Line= 2
2197519.66038681752704.1560217862197718.53511155752696.464734089
#Sta/Elev= 27
       0 1420.39     4.5 1420.33    14.9 1419.86    28.5 1418.91    32.5 1418.72
    40.5 1418.67    52.6 1418.29    60.6 1418.15    64.6 1417.53    68.6 1415.27
    72.51412.598    76.6 1411.34    80.6 1411.79   82.03 1412.58    83.81413.364
    84.6 1413.76    88.6 1416.61      89 1416.77    92.6  1418.1    96.6 1418.43
   120.6  1418.7   136.6 1418.52   148.6 1418.25   164.6 1418.22   172.6  1418.4
   180.6 1418.44     199 1418.73
#Mann= 5 ,-1,0
       0     .07       0      60     .06       0    72.5    .045       0
    83.8     .06       0     160     .05       0
Bank Sta=72.5,82.03
XS Rating Curve= 0 ,0
Exp/Cntr(USF)=0,0
Exp/Cntr=0.3,0.1

Type RM Length L Ch R = 1 ,249     ,46.9,46.5,46.1
XS GIS Cut Line= 2
2197525.70354143752738.2174387312197703.15253616752729.976773341
#Sta/Elev= 28
       0 1420.34    10.5 1419.99    14.8 1419.62    22.5 1418.81    26.7 1418.53
    35.1 1418.21    42.5 1418.08    50.5 1418.02    58.5 1418.11    62.5 1417.52
    66.61414.645   69.63 1412.27    70.5  1411.7    74.6 1411.21    78.6 1412.08
      791412.311    83.7 1415.01    86.6 1416.59    87.5 1416.95    90.6 1418.01
    94.6 1418.45   102.3 1418.53   118.2 1418.25   134.6 1418.36   146.6  1418.2
   158.6 1418.39   166.7  1418.4   177.6 1418.19
#Mann= 4 ,-1,0
       0     .07       0      60     .05       0    66.6    .045       0
      79     .05       0
Bank Sta=69.63,79
XS Rating Curve= 0 ,0
Exp/Cntr(USF)=0,0
Exp/Cntr=0.3,0.1

Type RM Length L Ch R = 1 ,203     ,161,161.7,161
XS GIS Cut Line= 2
2197480.20211413752791.368401942 2197769.1086677752767.289096365
#Sta/Elev= 30
       0    1419      16 1418.92    24.1  1418.6    60.2 1418.67   100.3 1417.61
   104.3 1417.19   105.7 1416.64   108.3 1415.48   112.4 1412.94114.96761411.671
   116.4 1410.97   120.4 1410.65128.36751411.805   132.4 1412.99   140.5 1416.51
   144.5 1417.54   148.5    1418   160.5 1418.25   172.6 1419.08   176.6 1418.61
   180.6 1418.41   208.7 1418.75   216.7  1418.5   220.6 1418.68   231.7 1418.52
   244.8 1418.78   248.8 1418.45   260.9  1418.9   264.9 1418.66   289.9 1418.82
#Mann= 4 ,-1,0
       0     .07       0     100     .05       0114.9676    .045       0
128.3675     .05       0
Bank Sta=114.9676,128.3675
XS Rating Curve= 0 ,0
Exp/Cntr(USF)=0,0
Exp/Cntr=0.3,0.1

Type RM Length L Ch R = 1 ,41      ,,,
XS GIS Cut Line= 4
2197478.19731154752949.6266257882197594.08544124752945.203414731
 2197667.5107448752933.7030659822197799.25698885  752919.7782358
#Sta/Elev= 30
       0 1419.84    17.8 1419.05      38 1418.59      54 1418.52      66  1418.7
      82 1418.15      98 1418.13   118.1 1418.54   124.8 1418.26   130.2 1417.88
   134.3 1416.99   138.3 1414.77   142.3 1411.69  145.13 1409.73   146.4 1408.94
   150.5 1408.62   152.8  1409.7   154.5 1410.49   158.6 1411.64   162.6 1413.06
   170.7 1416.34   174.8  1417.4   178.8 1417.96   186.9 1417.98   194.9 1418.34
   219.1  1418.8   243.3 1418.47   267.4  1418.4   299.6 1417.96   322.8 1418.23
#Mann= 5 ,-1,0
       0     .07       0  145.13    .045       0   152.8     .07       0
  200.29     .05       0  300.29     .06       0
Bank Sta=145.13,152.8
XS Rating Curve= 0 ,0
Exp/Cntr(USF)=0,0
Exp/Cntr=0.3,0.1
LCMann Table=0

Chan Stop Cuts=-1
Use User Specified Reach Order=0
Composite Channel Slope=5
